--- ANTHNYCK.prj (project) ---

Proj Title=ANTHNYCK
Current Plan=p01
Default Exp/Contr=0,0
English Units
Geom File=g01
Flow File=f01
Plan File=p01
Background Map Layer=Inundation Boundary (0_2pct Value_0)
Background Map Layer=Inundation Boundary (01pct Value_0)
BEGIN DESCRIPTION:
----------MODEL BY WOOD PLC 2021----------
Stream Name: Anthony Creek
Flood Zone: Enhanced Approximate
Pocahontas County, WV
HEC-RAS Version: RAS 6.1
Vertical Datum: NAVD88
Projection: NAD 1983 StatePlane West Virginia S FIPS 4702 (US Feet)
Terrain: 1-meter LIDAR (FEMA Region III 3DEP collected 2016-2018)
Land Use: 2019 NLCD
Hydrologic Method:
WV SIR2010-5033 regression equations
END DESCRIPTION:
DSS File=dss
DSS Export Rating Curves= 0
DSS Export Rating Curve Sorted= 0
DSS Export Volume Flow Curves= 0
DXF OffsetX= 0
DXF OffsetY= 0
DXF ScaleX= 0
DXF ScaleY= 0

--- ANTHNYCK.p01 (plan) ---

Plan Title=Floodplain
Program Version=6.10
Short Identifier=Floodplain
Geom File=g01
Flow File=f01
Subcritical Flow
K Sum by GR= 0
Std Step Tol= 0.01
Critical Tol= 0.01
Num of Std Step Trials= 20
Max Error Tol= 0.3
Flow Tol Ratio= 0.001
Split Flow NTrial= 30
Split Flow Tol= 0.02
Split Flow Ratio= 0.02
Log Output Level= 0
Friction Slope Method= 1
Unsteady Friction Slope Method= 2
Unsteady Bridges Friction Slope Method= 1
Parabolic Critical Depth
Global Vel Dist= 0 , 0 , 0
Global Log Level= 0
CheckData=True
Encroach Param=-1 ,0,0, 0
Computation Interval=0.1SEC
Output Interval=1SEC
Instantaneous Interval=Max Profile
Mapping Interval=1HOUR
Computation Time Step Use Courant=        0
Computation Time Step Use Time Series=    0
Computation Time Step Count To Double=0
Computation Time Step Max Doubling=0
Computation Time Step Max Halving=0
Computation Time Step Residence Courant=0
Run HTab= 0
Run UNet= 0
Run Sediment= 0
Run PostProcess= 0
Run WQNet= 0
Run RASMapper= 0
UNET Theta= 0
UNET Theta Warmup= 0
UNET ZTol= 0
UNET ZSATol= 0
UNET MxIter= 0
UNET Max Iter WO Improvement= 0
UNET MaxInSteps= 0
UNET DtIC= 0
UNET DtMin= 0
UNET MaxCRTS= 0
UNET WFStab= 0
UNET SFStab= 0
UNET WFX= 1
UNET SFX= 1
UNET Gravity=32.174
UNET 1D Methodology=Finite Difference
UNET DSS MLevel= 1
UNET Pardiso=0
UNET DZMax Abort= 0
UNET Use Existing IB Tables= 0
UNET Froude Reduction=False
UNET Froude Limit= 0
UNET Froude Power= 0
UNET D1 Cores= 0
UNET WindReference=Eulerian
UNET WindDragFormulation=Hsu (1988)
UNET D2 Coriolis=0
UNET D2 Cores= 0
UNET D2 Theta= 1
UNET D2 Theta Warmup= 1
UNET D2 Z Tol= 0.01
UNET D2 Volume Tol= 0.01
UNET D2 Max Iterations= 20
UNET D2 Equation= 0
UNET D2 RampUpFraction=0.1
UNET D2 TimeSlices= 1
UNET D2 Turbulence Formulation=Non-Conservative (original)
UNET D2 Eddy Viscosity=0.3
UNET D2 Transverse Eddy Viscosity=0.3
UNET D2 Smagorinsky Mixing=0
UNET D2 BCVolumeCheck=0
UNET D2 Cores=0
UNET D2 SolverType=PARDISO (Direct)
UNET D2 Minimum Iterations= 2147483647
UNET D2 Maximum Iterations= 2147483647
UNET D2 Restart Number= 10
UNET D2 Relaxation Coeff=1.3
UNET D2 SOR Precondition Iterations= 10
UNET D2 ILUT Maximum Fill= 8
UNET D2 ILUT Tolerance=1E-08
UNET D1D2 MaxIter= 0
UNET D1D2 ZTol=0.01
UNET D1D2 QTol=0.1
UNET D1D2 MinQTol=1
DSS File=dss
Write IC File= 0
Write IC File at Fixed DateTime=0
Write IC File at Sim End=0
Echo Input=False
Echo Parameters=False
Echo Output=False
Write Detailed= 0
HDF Write Warmup=0
HDF Write Time Slices=0
HDF Flush=0
HDF Compression= 1
HDF Chunk Size= 1
HDF Spatial Parts= 1
HDF Use Max Rows=0
HDF Fixed Rows= 1
Calibration Method= 0
Calibration Iterations= 20
Calibration Max Change=0.05
Calibration Tolerance=0.2
Calibration Maximum=1.5
Calibration Minimum=0.5
Calibration Optimization Method= 1
WQ AD Non Conservative
WQ ULTIMATE=-1
WQ Max Comp Step=1HOUR
WQ Output Interval=15MIN
WQ Output Selected Increments= 0
WQ Output face flow=0
WQ Output face velocity=0
WQ Output face area=0
WQ Output face dispersion=0
WQ Output cell volume=0
WQ Output cell surface area=0
WQ Output cell continuity=0
WQ Output cumulative cell continuity=0
WQ Output face conc=0
WQ Output face dconc_dx=0
WQ Output face courant=0
WQ Output face peclet=0
WQ Output face adv mass=0
WQ Output face disp mass=0
WQ Output cell mass=0
WQ Output cell source sink temp=0
WQ Output nsm pathways=0
WQ Output nsm derived pathways=0
WQ Create Restart=0
WQ Fixed Restart=0
WQ System Summary=0
WQ Write To DSS=0
Sorting and Armoring Iterations= 10
XS Update Threshold= 0.02
Bed Roughness Predictor= 0
Hydraulics Update Threshold= 0.02
Energy Slope Method= 1
Volume Change Method= 1
Sediment Retention Method= 0
Sediment TS Multiplier= 1
Warm Up Method= 0
XS Weighting Method= 0
Number of US Weighted Cross Sections= 1
Number of DS Weighted Cross Sections= 1
Upstream XS Weight=0
Main XS Weight=1
Downstream XS Weight=0
Number of DS XS's Weighted with US Boundary= 1
Upstream Boundary Weight= 1
Weight of XSs Associated with US Boundary= 0
Number of US XS's Weighted with DS Boundary= 1
Downstream Boundary Weight= 0.5
Weight of XSs Associated with DS Boundary= 0.5
Percentile Method= 0
Sediment Output Level= 3
Mass or Volume Output= 0
Output Increment Type= 1
Profile and TS Output Increment= 1
Transport Output Increment 1
XS Output Flag= 0
XS Output Increment= 10
Read HDF5 Sediment Hotstart= 0
Sediment Hotstart Type= 0
Write Gradation File= 0
Read Gradation Hotstart= 0
Write HDF5 File= 1
Write Binary Output= 1
Write DSS Sediment File= 0
DSS Sediment Output Type= 1
SV Curve= 0
Specific Gage Flag= 0
Subcell Erosion Methods= 0
Subcell Deposition Methods= 0
Advection Scheme= 1
Matrix Solver= 0
Implicit Weighting Factor= 1
Maximum Outer Loop Convergence Iterations= 5
Convergence Maximum Absolute= 0.001
Convergence RMSE= 0.0001
Grain Fractions Max Abs Error= 0.001
Max Subgrid Regions= 1
Max Subgrid Length Scale= 3.402823E+38
Initial Layer Thickness= 3.402823E+38
Min Layer Thickness= 3.402823E+38
Max Layer Thickness= 3.402823E+38
Number of Layers= 5

--- ANTHNYCK.f01 (steady flow) ---

Flow Title=Flow
Program Version=6.00
Number of Profiles= 6
Profile Names=01pct,10pct,04pct,02pct,0_2pct,01plus
River Rch & RM=ANTHNYCK,Main            ,10209
     709     378     501     601     987    1050
River Rch & RM=ANTHNYCK,Main            ,8414
     806     432     575     685    1120    1190
River Rch & RM=ANTHNYCK,Main            ,7226
     909     489     644     772    1260    1340
River Rch & RM=ANTHNYCK,Main            ,3358
    1060     573     754     902    1460    1570
River Rch & RM=ANTHNYCK,Main            ,2678
    1310     714     935    1120    1800    1930
Boundary for River Rch & Prof#=ANTHNYCK,Main            , 1
Up Type= 0
Dn Type= 1
Dn Known WS=2334.3
Boundary for River Rch & Prof#=ANTHNYCK,Main            , 2
Up Type= 0
Dn Type= 1
Dn Known WS=2333.1
Boundary for River Rch & Prof#=ANTHNYCK,Main            , 3
Up Type= 0
Dn Type= 1
Dn Known WS=2333.6
Boundary for River Rch & Prof#=ANTHNYCK,Main            , 4
Up Type= 0
Dn Type= 1
Dn Known WS=2333.9
Boundary for River Rch & Prof#=ANTHNYCK,Main            , 5
Up Type= 0
Dn Type= 1
Dn Known WS=2335.1
Boundary for River Rch & Prof#=ANTHNYCK,Main            , 6
Up Type= 0
Dn Type= 1
Dn Known WS=2335.3
DSS Import GetInterval= 0
DSS Import GetPeak= 0
DSS Import FillOption= 0

--- ANTHNYCK.g01 (geometry) ---

Geom Title=Geometry
Program Version=6.10

River Reach=ANTHNYCK        ,Main
Reach XY= 30
     2258295.195      394626.533     2258329.019      394538.633
     2258057.469       394578.27     2257952.318      394456.744
     2257666.481      394626.504     2257459.061      394616.418
     2257213.973      394409.918     2257126.733      393997.975
     2256547.914      394005.665     2256368.862      393732.273
     2256331.698      393546.372     2256369.867      393187.068
     2256287.188      392489.858     2256105.174      392255.374
     2255972.313      391892.983     2255395.974      390860.447
     2255413.858      390352.491     2254924.773      390075.548
2254867.06446553390084.581494396     2254851.294      390193.019
2254756.50075458390208.278754576     2254410.871390017.837037675
     2254392.185      389831.237     2254489.554      389408.432
     2254946.217      388997.413     2254988.493      388678.082
     2255121.255      388464.539     2255094.852      388362.531
2254894.20744867388278.295222033      2254858.48      388058.511

Type RM Length L Ch R = 1 ,10209   ,408,408,408
XS GIS Cut Line= 4
 2258685.4316933      394558.6412258426.01903094394556.541419665
2258106.70758185 394719.46721302     2258003.071      395057.778
#Sta/Elev= 30
       0 2494.05     5.3 2492.24    13.3 2487.81    29.3 2486.59    41.3 2480.88
    85.3 2466.25   169.3 2435.99   193.3  2428.8   229.3 2424.13   260.8 2422.09
   301.9 2421.21   338.6 2418.49   362.4 2419.52   395.1 2419.24   412.9  2418.3
   421.8 2419.58     477 2418.48   542.5 2421.05   568.9 2420.53   666.1 2422.18
   774.5 2426.49   795.4  2431.8   807.9 2433.51   841.4 2434.22   849.8 2438.68
   858.1 2445.56   867.9 2449.89   880.7 2453.21   899.9 2459.95   971.7 2476.16
#Mann= 10 ,-1,0
       0      .1       0  359.42     .05       0  389.42      .1       0
   395.1    .045       0   421.8      .1       0  499.42     .05       0
  609.42     .06       0   707.9     .07       0   807.9     .06       0
   907.9      .1       0
Bank Sta=395.1,421.8
XS Rating Curve= 0 ,0
Exp/Cntr=0.3,0.1

Type RM Length L Ch R = 1 ,9801    ,367.4,353.4,327.8
XS GIS Cut Line= 3
2258140.32343347394230.5719567882258024.87229416394719.019084643
2257882.77858424394978.784148094
#Sta/Elev= 30
       0 2517.03    43.8 2509.33    55.5 2506.41    88.7 2496.14   121.9 2483.31
   150.6    2471   171.2 2459.32   187.6 2451.28   226.7 2434.22   232.9 2430.79
   249.3 2417.96   265.7 2416.31   335.6  2416.2  342.48 2414.48   347.9 2413.59
   363.9 2413.56   372.6 2414.34     389 2416.31   409.6 2415.92   431.1 2419.26
   451.1 2420.29   604.7 2422.81   610.1 2423.47   621.9 2429.17   627.5 2430.06
   686.8 2428.88   691.3 2429.94   695.1 2431.84   716.2 2444.59     798 2479.24
#Mann= 8 ,-1,0
       0      .1       0  342.48    .045       0   372.6      .1       0
     380     .05       0     490     .06       0  511.91     .08       0
  591.91     .06       0  711.91      .1       0
Bank Sta=342.48,372.6
XS Rating Curve= 0 ,0
Exp/Cntr(USF)=0,0
Exp/Cntr=0.3,0.1

Type RM Length L Ch R = 1 ,9447    ,96.2,91,84.8
XS GIS Cut Line= 4
2257739.92578308394140.100854162 2257727.4871175 394414.93613158
2257859.42582019394616.1759710252257836.76967932394973.343368187
#Sta/Elev= 30
       0 2506.43    17.1 2500.73    41.1 2490.51    69.1 2480.05    97.2 2470.73
   121.2  2461.3   157.2 2442.26   181.7  2424.3   193.3 2416.61   197.3 2414.93
   205.3 2413.92   294.4 2412.12   411.7 2414.05   416.5 2412.32   421.3 2410.21
   424.6 2410.06   440.4 2412.23   453.5  2414.6   464.3  2413.9   483.5 2415.17
   580.9  2417.5   604.9 2420.48   629.1 2425.41     649 2425.82   709.1 2424.36
   721.2 2425.33   741.2 2425.17     761 2431.48   781.3  2439.8 873.637 2483.99
#Mann= 10 ,-1,0
       0      .1       0     170     .07       0     270     .06       0
  385.12     .05       0   416.5    .045       0   440.4     .05       0
  455.12      .1       0  505.12     .08       0  605.75     .07       0
  705.75      .1       0
#XS Ineff= 2 , 0
          392.87 2429.85
Permanent Ineff=
       F       F
Bank Sta=416.5,440.4
XS Rating Curve= 0 ,0
Exp/Cntr(USF)=0,0
Exp/Cntr=0.5,0.3

Type RM Length L Ch R = 1 ,9356    ,82.7,77.5,74.5
XS GIS Cut Line= 4
2257697.75100246394067.5774266962257575.83490684394448.849709026
2257821.31677821394668.4208089652257794.87897867 394965.14815153
#Sta/Elev= 30
       0 2514.28      28  2508.6    52.1 2500.45   110.9 2477.19   148.7  2460.2
   173.9 2447.91   209.9 2418.43   215.7  2414.5   222.1 2412.36   420.6 2410.53
   465.9 2412.45   490.8 2410.67   570.7  2414.6   598.8 2413.72   602.82411.057
     610 2409.56   627.4 2411.12   634.8 2413.88   642.2 2414.87   658.8 2414.12
   678.4 2416.71   701.3 2415.27   738.8 2416.96   746.5 2418.76   754.5 2422.65
   762.5 2424.08   886.3  2423.2   912.1  2431.1   931.2 2438.44  1027.5 2485.45
#Mann= 8 ,-1,0
       0      .1       0     240     .06       0  470.29     .07       0
  480.29     .06       0   602.8    .045       0   627.4     .05       0
  630.29     .06       0  859.64      .1       0
#XS Ineff= 2 , 0
           571.7  2418.6  638.61          2420.7
Permanent Ineff=
       F       F
Bank Sta=602.8,627.4
XS Rating Curve= 0 ,0
Exp/Cntr=0.5,0.3

Type RM Length L Ch R = 1 ,9279    ,176.3,203.4,232
XS GIS Cut Line= 4
2257663.79404196394054.3663151462257509.19919842394491.496562418
 2257763.7476046394711.2571306642257741.09146374394945.952093882
#Sta/Elev= 30
       0  2511.1    24.2 2503.85    96.3 2474.46   130.4 2459.39     160 2444.12
   193.1 2420.87   205.6    2413   210.9 2411.03   313.8 2410.49   343.5  2411.4
   381.2 2410.11   389.1 2410.56     406 2414.33   430.7  2415.9   444.2 2409.87
   448.5 2409.49   594.6 2411.63   625.4 2413.82   651.3 2410.72   665.5 2409.02
   692.7 2410.77   699.5  2413.6     705  2414.4   833.7 2417.65   870.2 2422.29
   886.3 2422.04   894.3 2424.85   918.6 2430.45   962.6 2445.621035.736  2479.7
#Mann= 7 ,-1,0
       0      .1       0     170     .06       0  483.66      .1       0
  493.66     .06       0   651.3    .045       0   692.7     .06       0
  889.95      .1       0
#XS Ineff= 2 , 0
           648.5  2418.6   693.8          2420.7
Permanent Ineff=
       F       F
Bank Sta=651.3,692.7
XS Rating Curve= 0 ,0
Exp/Cntr(USF)=0,0
Exp/Cntr=0.5,0.3

Type RM Length L Ch R = 1 ,9075    ,281.6,312.1,336.2
XS GIS Cut Line= 3
2257625.72241642394050.8327706932257488.31574655394400.111743113
2257438.01447036394874.592721767
#Sta/Elev= 30
       0 2500.87    62.7  2474.4   101.7 2456.13   132.6  2440.2   175.8 2414.17
   181.9 2411.77     190 2410.41   200.2 2409.75   316.3 2410.37   342.9 2409.33
   350.7 2409.72   363.9 2413.25   396.5 2415.55   401.9 2415.09   416.4 2410.17
   432.7 2408.94   521.2  2410.6   533.3 2409.37   578.9 2409.23   598.3 2407.61
   609.2 2408.33  611.18 2409.28   617.8 2413.84   625.8 2420.94   629.8  2423.2
   649.9 2424.48     662 2431.61   706.2  2450.1   799.3 2483.68852.4749 2501.96
#Mann= 7 ,-1,0
       0      .1       0     170     .06       0     270     .07       0
     280     .06       0  485.34      .1       0   578.9    .045       0
  611.18      .1       0
#XS Ineff= 2 , 0
           398.3 2437.35
Permanent Ineff=
       F       F
Bank Sta=578.9,611.18
XS Rating Curve= 0 ,0
Exp/Cntr(USF)=0,0
Exp/Cntr=0.3,0.1

Type RM Length L Ch R = 1 ,8763    ,269.7,276.2,272.8
XS GIS Cut Line= 4
2257604.58787881394010.3072423822257420.38009288394346.925781857
2257122.19454776394475.4701627082257099.85344278394608.385587474
#Sta/Elev= 30
       0 2505.33    35.2 2490.28    64.3 2475.82   111.5 2450.37   155.7 2422.28
     172 2413.42   182.2 2410.32     194 2409.31   325.8 2408.63   342.5 2409.38
   356.1 2413.75   381.7 2415.56     397 2408.61   409.9 2407.65   452.6 2407.75
   484.1 2405.53   492.8  2406.9     553 2408.09   581.4 2406.39     593 2404.33
  603.82 2406.46   621.8  2410.8   649.7 2414.53   675.8 2413.64   684.5 2416.63
   708.4 2420.99   753.3 2436.89   787.2 2446.19   812.4 2450.68   843.2 2451.72
#Mann= 6 ,-1,0
       0      .1       0     230     .07       0     340     .06       0
     370      .1       0   581.4    .045       0  603.82      .1       0
#XS Ineff= 2 , 0
          380.34 2416.73
Permanent Ineff=
       F       F
Bank Sta=581.4,603.82
XS Rating Curve= 0 ,0
Exp/Cntr=0.3,0.1

Type RM Length L Ch R = 1 ,8414    ,210.6,193.3,169.9
XS GIS Cut Line= 3
2257539.45922967394042.6085673772257066.58366533394222.684712954
 2256954.7739344394549.464842852
#Sta/Elev= 30
       0  2470.5    29.3 2455.01    37.8 2451.64    59.2 2440.06    84.8 2424.48
   106.8 2412.99   119.2  2408.3   131.6 2407.16   165.7 2407.74   187.9 2406.46
   226.1 2406.17   233.9 2407.38   247.5 2414.27   271.1 2415.98     330 2406.27
   350.2 2404.57   358.8 2402.28   363.1 2401.18   375.9 2400.86   382.7 2402.18
   388.7 2403.75   410.1 2404.72   601.6 2408.67   622.8 2408.04   642.2 2409.89
   736.7 2412.83   783.4 2419.71   817.3 2422.03   825.7 2421.77   851.4 2424.12
#Mann= 7 ,-1,0
       0      .1       0     120     .06       0     190      .1       0
     230     .07       0     330      .1       0   358.8    .045       0
   382.7      .1       0
#XS Ineff= 2 , 0
          269.98 2416.11
Permanent Ineff=
       F       F
Bank Sta=358.8,382.7
XS Rating Curve= 0 ,0
Exp/Cntr=0.3,0.1

Type RM Length L Ch R = 1 ,8293    ,238.9,241.5,241.3
XS GIS Cut Line= 2
 2257179.7158721393846.1783730752256965.70942367 394463.02048913
#Sta/Elev= 30
       0 2417.03    20.9 2416.84      37 2412.63    66.7 2411.68    87.9 2410.16
   105.7 2407.73   121.4 2403.22   130.2 2402.26   138.7 2402.97     145 2402.72
   147.1 2402.47  153.04 2400.15   155.6 2399.06   159.2 2398.87   169.4 2400.06
   176.8 2401.99   203.2 2401.73   219.1 2403.54   271.4 2403.64     325 2405.64
   392.7 2407.17     440 2407.17   486.1 2408.52     507  2408.5   536.6 2409.66
   570.9 2409.94   583.5 2411.52   600.2 2411.22   612.9 2412.84   652.9 2414.36
#Mann= 6 ,-1,0
       0     .06       0  153.04    .045       0   169.4     .06       0
     180      .1       0     440     .06       0     490      .1       0
#XS Ineff= 2 , 0
                          259.51         2406.95
Permanent Ineff=
       F       F
Bank Sta=153.04,169.4
XS Rating Curve= 0 ,0
Exp/Cntr(USF)=0,0
Exp/Cntr=0.3,0.1

Type RM Length L Ch R = 1 ,8052    ,345.3,352.4,353.5
XS GIS Cut Line= 4
2257159.58638925  393749.97554972256935.78879613393917.823744545
2256849.86650591394125.6357953052256764.83598116394417.761107521
#Sta/Elev= 30
       0 2417.18    19.3  2417.3    33.3 2414.53     152 2411.35   219.3 2407.57
   244.7 2404.59   259.3 2402.14   274.3 2400.86   320.6 2400.71   337.1 2401.57
   343.3 2400.54   353.1 2397.65   361.6 2396.46   370.8 2397.55   382.9 2400.98
   391.6 2401.83   446.2 2402.01   467.2 2403.48   545.8 2405.66   591.6 2407.99
     600 2409.81   616.6 2416.09   657.3 2435.38     675 2442.41   699.9 2450.87
   724.9 2457.78   749.9 2462.52   774.9 2465.35   792.8 2465.27   808.9 2463.12
#Mann= 9 ,-1,0
       0     .07       0     110     .06       0     160     .07       0
     270     .06       0  279.75      .1       0   353.1    .045       0
   370.8      .1       0  544.62     .07       0  594.62      .1       0
#XS Ineff= 2 , 0
           335.6 2403.83  393.19         2402.51
Permanent Ineff=
       F       F
Bank Sta=353.1,370.8
XS Rating Curve= 0 ,0
Exp/Cntr(USF)=0,0
Exp/Cntr=0.3,0.1

Type RM Length L Ch R = 1 ,7700    ,453.8,473.4,488.4
XS GIS Cut Line= 3
2257048.00828059393690.814661616 2256752.9325486393764.971492431
2256432.39863283394232.790386603
#Sta/Elev= 30
       0 2411.54   160.7 2407.56   186.4 2405.14   251.4 2401.59   304.3 2402.22
   367.5    2399   435.4 2397.69   440.1 2397.24     450  2394.5   475.4 2392.71
     492 2393.55   517.9 2393.47   546.6 2395.11   551.8 2396.28   556.6 2398.82
   561.5 2400.22   566.3 2399.57   584.1 2394.63   609.9 2394.16   624.3 2393.15
     633 2394.52   639.1 2398.61   653.1 2412.45     656  2414.1   680.7 2422.45
   696.3 2428.56   776.8 2465.15   808.8 2476.74   842.7 2483.71   871.3 2487.65
#Mann= 6 ,-1,0
       0     .06       0     100     .07       0  334.25     .06       0
  364.25      .1       0   609.9    .045       0     633      .1       0
#XS Ineff= 2 , 0
           562.3    2412
Permanent Ineff=
       F       F
Bank Sta=609.9,633
XS Rating Curve= 0 ,0
Exp/Cntr=0.3,0.1

Type RM Length L Ch R = 1 ,7226    ,171.2,172.9,174.3
XS GIS Cut Line= 3
2257005.58383154393464.7541317512256621.87779051393583.005086392
2256120.86607128393664.388151187
#Sta/Elev= 30
       0 2407.85    68.4 2403.99   148.6 2403.68   189.8 2402.87   202.4 2401.93
   294.5  2399.1   549.1 2394.05   581.5 2394.25   593.1 2390.88   613.8 2388.64
     642 2388.61   650.4 2389.38   664.5 2387.93   670.7 2387.29   686.4 2387.93
   690.8 2388.75   701.2 2394.35   707.2  2395.6   739.6 2395.78   747.7 2396.74
   755.8 2393.07   759.9 2393.76   763.9 2395.84   776.1 2399.01   784.2 2404.21
   804.4 2419.59     845 2444.12   875.5 2463.94   889.5 2471.89   909.1 2485.08
#Mann= 6 ,-1,0
       0     .05       0      80     .06       0     380     .05       0
  481.51      .1       0   664.5    .045       0   686.4      .1       0
#XS Ineff= 2 , 0
           649.9 2394.94
Permanent Ineff=
       F       F
Bank Sta=664.5,686.4
XS Rating Curve= 0 ,0
Exp/Cntr=0.3,0.1

Type RM Length L Ch R = 1 ,7053    ,259.8,262.1,263.6
XS GIS Cut Line= 2
 2257018.4343669 393396.757741062256138.26713937393472.896774583
#Sta/Elev= 30
       0 2415.22    10.3 2410.27    30.4 2408.17    74.5 2405.77   134.8 2403.97
   168.8 2401.52   227.1 2400.59   347.6  2396.7   395.7 2396.31     480 2393.02
   620.6 2393.01   652.7 2390.56   664.7 2388.61   676.8 2388.29   685.52386.438
   700.9 2385.81   706.6 2386.33   712.9 2387.33   716.9  2390.8   720.9 2392.35
     741 2392.28     749 2393.72   781.2 2393.02     797 2394.23   809.3 2396.93
   813.3 2398.61   829.3 2410.51   854.7 2430.29   873.5 2446.79   883.5 2453.74
#Mann= 6 ,-1,0
       0     .07       0     180     .06       0     280     .05       0
     480      .1       0   685.5    .045       0   706.6      .1       0
Bank Sta=685.5,706.6
XS Rating Curve= 0 ,0
Exp/Cntr(USF)=0,0
Exp/Cntr=0.3,0.1

Type RM Length L Ch R = 1 ,6791    ,355.8,356.1,355.3
XS GIS Cut Line= 3
2256889.53800216393151.4653714932256583.43733262393204.624611234
2256129.20548309393203.042500639
#Sta/Elev= 30
       0 2415.32    25.7 2415.52      42 2414.19    86.6 2408.67   119.1 2402.36
   147.9 2398.36   171.9 2397.63   204.4 2395.26   220.6 2395.44     260 2393.85
   277.5 2393.42   309.9 2390.05   417.9 2388.72   457.9 2386.98   497.9 2387.34
   509.9 2386.63   516.7 2384.41   521.9 2383.62   536.6 2384.25   545.9 2385.08
   565.9 2384.16   573.9 2389.23   577.9 2390.61   589.9 2390.17   597.9 2386.53
   609.9 2388.44   623.6 2392.91   637.9 2401.84   681.9 2438.85   764.9  2501.2
#Mann= 6 ,-1,0
       0     .05       0      60     .08       0     260     .05       0
  350.68      .1       0   516.7    .045       0   536.6      .1       0
#XS Ineff= 2 , 0
                          583.12         2402.29
Permanent Ineff=
       F       F
Bank Sta=516.7,536.6
XS Rating Curve= 0 ,0
Exp/Cntr=0.3,0.1

Type RM Length L Ch R = 1 ,6435    ,246.3,238.7,231
XS GIS Cut Line= 4
2256880.57726686392947.8879168032256699.54151071392843.437203811
2256256.62779139392852.7690340812256144.02892406392885.185069125
#Sta/Elev= 30
       0 2407.29    14.3  2407.1    22.8 2406.23    51.3 2400.58    92.8    2391
   111.3 2388.23   128.2 2387.26   236.4 2386.07   260.4 2385.09   276.4 2385.25
   292.4 2386.34   312.8 2384.75   484.4 2382.66   500.4 2383.61   528.4 2382.64
   540.4  2383.8   548.4 2381.72   556.5 2380.69   572.5 2380.53   576.5 2380.59
   580.5 2381.76   584.5 2385.06   588.5 2386.11   620.5 2387.86   624.5 2388.61
   636.5 2392.88   652.5 2400.86   711.3 2439.52   735.7 2454.04   769.2 2470.96
#Mann= 7 ,-1,0
       0     .07       0      50      .1       0     170     .05       0
  269.01     .06       0  369.01      .1       0   548.4    .045       0
   580.5      .1       0
#XS Ineff= 2 , 0
          419.28  2399.1
Permanent Ineff=
       F       F
Bank Sta=548.4,580.5
XS Rating Curve= 0 ,0
Exp/Cntr=0.3,0.1

Type RM Length L Ch R = 1 ,6196    ,32.1,33.5,35.2
XS GIS Cut Line= 2
2256754.22825596392491.955508647 2256038.9741554392692.191681054
#Sta/Elev= 30
       0 2391.84    10.4 2390.93    18.7 2387.08    22.9 2385.99    60.3  2384.1
   122.3 2382.62     160 2382.33   207.1  2382.4   220.1 2383.27   238.9 2384.27
   265.5 2382.46   326.1 2381.41   411.6 2382.22     430 2380.95   442.4  2378.9
   447.3 2377.85   454.9 2377.62   468.5 2378.96   492.3 2383.67   546.3 2384.55
   568.4 2384.15   583.6 2385.43   600.3 2388.86   604.4 2390.32   612.7 2395.05
     621 2398.79   704.1 2444.32   712.4  2449.4     729 2457.84742.7536 2462.04
#Mann= 6 ,-1,0
       0     .06       0   122.3     .05       0     160     .06       0
   220.1      .1       0   442.4    .045       0   468.5      .1       0
#XS Ineff= 2 , 0
             400  2408.3  494.79         2401.51
Permanent Ineff=
       F       F
Bank Sta=442.4,468.5
XS Rating Curve= 0 ,0
Exp/Cntr(USF)=0,0
Exp/Cntr=0.5,0.3

Type RM Length L Ch R = 1 ,6163    ,29.7,29.9,30.1
XS GIS Cut Line= 3
2256740.23795571392458.7285455412256417.58665607392557.535041095
2256023.23506761392645.848811457
#Sta/Elev= 30
       0 2390.45     5.2 2390.06    12.6 2386.69    16.8 2385.33    37.7 2384.54
   130.1 2382.72   175.8 2382.52   234.3 2383.77   242.7 2382.78     272 2382.56
   392.2 2383.82   416.8 2381.76   433.2 2378.96   437.3 2378.03   445.4 2377.56
   458.9 2378.87     466 2378.93   470.1 2380.21   474.2 2382.67   478.3 2383.53
   584.8 2384.06   592.9 2384.34   599.6 2385.49   609.6 2388.68     625 2395.78
     690 2431.54     700 2438.32   711.9 2444.29   720.1 2447.37741.5607 2451.57
#Mann= 6 ,-1,0
       0     .06       0     110     .05       0     210     .06       0
     260      .1       0   433.2    .045       0   458.9      .1       0
#XS Ineff= 4 ,-1
       0     234    2390     234     410  2382.3     480     513  2383.5
     513     600    2390
Permanent Ineff=
       F       F       F       F
Bank Sta=433.2,458.9
XS Rating Curve= 0 ,0
Exp/Cntr(USF)=0,0
Exp/Cntr=0.5,0.3

Type RM Length L Ch R = 1 ,6133    ,64.5,61.8,59.7
XS GIS Cut Line= 3
2256727.99644298392425.5015824342256413.21468724392528.680046818
2256022.36067385392613.496242117
#Sta/Elev= 30
       0 2389.23       4 2388.87    12.4 2385.41    20.9 2384.64    50.3 2383.62
   196.2 2381.88   214.5 2382.08     231 2382.97   240.5 2381.85     332 2383.06
   389.6 2383.16   396.5 2382.91   414.2 2381.08   430.1 2378.49   434.7 2377.56
   443.5  2377.4   450.3 2377.73   455.1 2378.67   463.3 2378.92   467.4 2381.62
   470.4 2382.87   475.6 2383.69   553.4 2383.15   598.4    2384   606.6 2385.06
   619.5 2390.34   672.2 2418.94   704.8 2434.96   721.2 2439.77731.2111 2441.63
#Mann= 6 ,-1,0
       0     .06       0      90     .05       0     200     .06       0
     300      .1       0   430.1    .045       0   455.1      .1       0
#XS Ineff= 4 ,-1
      33     232    2390     232     414    2382     467     484    2383
     484     600    2390
Permanent Ineff=
       F       F       F       F
Bank Sta=430.1,455.1
XS Rating Curve= 0 ,0
Exp/Cntr(USF)=0,0
Exp/Cntr=0.5,0.3

Type RM Length L Ch R = 1 ,6071    ,210.3,202.3,194.7
XS GIS Cut Line= 2
 2256709.6341739392361.6708375182256014.49112995392577.646097712
#Sta/Elev= 30
       0 2387.45     5.7 2386.99    14.1 2382.76    18.3 2381.55    51.8 2380.72
    96.6 2381.57   202.1 2380.92   231.9 2381.68     241 2380.67   307.3 2382.05
     413 2382.29   416.3 2382.17  426.38 2378.45   428.8 2377.28     433 2376.79
   445.5 2376.95   453.9 2378.29   462.3  2378.1   470.7 2380.91     479 2380.86
   487.4  2382.8   525.1 2382.65   582.4 2383.58   611.2 2385.51   620.7 2388.81
   643.1 2399.41   692.6 2421.16   710.2 2426.14     722 2428.49727.9211 2429.01
#Mann= 4 ,-1,0
       0     .06       0     280      .1       0  426.38    .045       0
   453.9      .1       0
#XS Ineff= 2 , 0
          392.45 2394.81
Permanent Ineff=
       F       F
Bank Sta=426.38,453.9
XS Rating Curve= 0 ,0
Exp/Cntr(USF)=0,0
Exp/Cntr=0.3,0.1

Type RM Length L Ch R = 1 ,5869    ,500.5,503.7,504
XS GIS Cut Line= 4
2256641.15227428392124.9416059542256381.43368817       392190.05
2256061.80162621392403.8804163962255962.34029164392600.323690649
#Sta/Elev= 30
       0 2384.39    17.5 2382.69    25.8 2377.85    29.9 2377.34      34 2378.03
   126.3 2378.68   202.1 2378.52   236.1  2379.2   283.7 2378.58   341.5 2379.61
   375.1 2379.22   461.8 2380.19   489.2 2379.41   500.3 2376.29   510.8 2376.47
     516 2375.78   524.7 2374.68   538.8 2375.68   546.7 2380.88   548.4 2381.28
   562.8  2382.9   572.5 2383.02   582.3 2384.86   597.1 2386.36   625.9 2387.94
   653.8 2391.11   682.5 2396.41   774.8 2409.89   837.6 2422.29   872.5 2427.09
#Mann= 8 ,-1,0
       0     .06       0      60     .05       0     100     .07       0
     210     .06       0  317.76     .07       0  357.76      .1       0
     516    .045       0   538.8      .1       0
#XS Ineff= 2 , 0
          413.21 2394.67
Permanent Ineff=
       F       F
Bank Sta=516,538.8
XS Rating Curve= 0 ,0
Exp/Cntr=0.3,0.1

Type RM Length L Ch R = 1 ,5365    ,291.2,291.5,291.8
XS GIS Cut Line= 3
2256419.78738558391634.7815895042255762.44004991392007.155505666
2255746.31179126  392138.5784697
#Sta/Elev= 30
       0 2380.37    13.2 2380.59    21.1 2379.88    33.8 2373.64    36.3 2372.65
    39.6 2372.42    45.5 2372.75    51.4 2373.91    63.9 2374.41   247.8 2375.28
   297.9 2374.73   381.1  2375.5   482.3 2377.83   486.9 2377.29   500.4 2372.26
   505.2 2371.24   509.8 2369.58     519 2369.22   523.6 2369.84   526.8 2371.13
     542 2378.34   551.2 2379.67   569.6 2380.83   702.9 2384.84   720.5 2386.13
   739.7 2388.77   761.6 2393.32   777.7 2398.69     818 2409.99   887.9 2431.13
#Mann= 8 ,-1,0
       0     .06       0     200     .07       0     230     .06       0
     310     .07       0     430     .12       0   505.2    .045       0
   526.8     .12       0     630      .1       0
#XS Ineff= 2 , 0
          480.19 2398.13
Permanent Ineff=
       F       F
Bank Sta=505.2,526.8
XS Rating Curve= 0 ,0
Exp/Cntr=0.3,0.1

Type RM Length L Ch R = 1 ,5074    ,31.1,31.1,31.3
XS GIS Cut Line= 3
 2256279.7445327391385.9918535772255662.81115338391726.033873674
2255552.05460969391760.038075684
#Sta/Elev= 30
       0  2379.6     8.6 2378.68    17.8 2374.01    22.6  2372.4   180.6 2370.74
   231.7  2371.7     267    2371   405.4 2372.38   487.2  2373.9   492.8 2373.51
   499.6 2369.74   499.6 2369.73   502.6 2367.79   505.5 2366.85   511.1 2366.65
   520.3 2366.85   526.1 2369.38   529.1 2370.68   536.9 2375.75   540.9 2376.56
   675.5 2379.19   693.7 2380.02   705.9 2382.09   715.7 2387.58   728.3 2393.09
   744.9 2404.68   753.9 2409.54     770 2421.24   790.9 2439.83820.2987 2457.35
#Mann= 10 ,-1,0
       0     .06       0     140     .05       0     150     .06       0
     340     .05       0     380     .06       0   499.6    .045       0
   526.1     .06       0     550     .05       0     600     .06       0
  714.44      .1       0
#XS Ineff= 2 , 0
          477.36 2399.72
Permanent Ineff=
       F       F
Bank Sta=499.6,526.1
XS Rating Curve= 0 ,0
Exp/Cntr(USF)=0,0
Exp/Cntr=0.5,0.3

Type RM Length L Ch R = 1 ,5043    ,33.2,33,32.9
XS GIS Cut Line= 3
2256265.75566659391360.2521544862255660.29289933391691.251461213
2255532.50454429391735.084514917
#Sta/Elev= 30
       0 2379.42     6.4 2378.88    18.6 2372.92    24.6 2372.19    34.3 2372.58
    72.6 2371.58   184.6  2370.5   234.3  2371.5   252.5 2370.51   421.2 2371.98
     485 2373.13   494.1 2373.84   498.7 2373.32   504.5  2369.3   510.6 2366.87
   516.9 2366.51   521.5 2366.91   524.6 2369.39   530.6 2374.66   541.2  2375.8
     558 2376.61   676.5 2378.55   694.4 2380.56   698.6 2381.87   707.1 2387.95
   715.5 2396.51   732.4 2409.89   774.7 2436.62   796.5 2448.73825.1301 2463.17
#Mann= 4 ,-1,0
       0     .06       0   504.5    .045       0   524.6     .06       0
  700.03      .1       0
#XS Ineff= 2 , 0
          488.86  2375.4  536.43          2376.4
Permanent Ineff=
       F       F
Bank Sta=504.5,524.6
XS Rating Curve= 0 ,0
Exp/Cntr(USF)=0,0
Exp/Cntr=0.5,0.3

Type RM Length L Ch R = 1 ,5010    ,65.8,66,66.5
XS GIS Cut Line= 4
2256252.87968138391343.3206695622256021.87589217391454.380183605
2255656.75160458391656.5467726422255520.46536927391703.409370407
#Sta/Elev= 30
       0 2378.99     5.2 2377.71    13.9 2372.46    18.5 2372.22   187.2 2370.29
   214.7 2370.58   227.1 2371.32   271.4  2370.8   377.7 2371.05   486.9 2373.51
   492.1 2373.14   503.9 2369.15   509.7 2366.32   514.3 2366.15   518.9 2366.74
   523.4  2369.4   530.4 2373.81   536.2 2375.26   592.2 2375.81   637.8 2377.47
     656 2377.33   671.6 2378.43   674.3 2379.54   678.5  2382.4   687.2 2390.46
   695.4 2396.49   733.5 2420.26   761.7 2435.33     780 2443.85817.7896 2460.07
#Mann= 6 ,-1,0
       0     .06       0     230     .05       0     250     .06       0
   503.9    .045       0   523.4     .06       0  673.67      .1       0
#XS Ineff= 2 , 0
          496.57  2375.4  527.39          2376.4
Permanent Ineff=
       F       F
Bank Sta=503.9,523.4
XS Rating Curve= 0 ,0
Exp/Cntr(USF)=0,0
Exp/Cntr=0.5,0.3

Type RM Length L Ch R = 1 ,4944    ,284,285.6,286.6
XS GIS Cut Line= 3
 2256222.4231636 391282.036150292255648.23792395391582.244676604
2255508.33492139391624.021267645
#Sta/Elev= 30
       0 2378.66     7.1 2377.43    12.9  2373.9    16.1 2372.47    83.8 2370.79
   201.1 2369.53   214.7 2369.67   228.2 2370.57   241.8 2369.31   286.9 2369.82
   381.7 2369.73   485.5 2371.28   490.1 2371.05   499.2 2368.18   507.5 2365.96
   512.6 2365.74   517.1 2365.88   522.7 2368.12   530.6 2372.16   537.5 2372.96
   608.7 2375.94   634.5 2377.38     639 2378.46   644.2 2380.54   652.2 2382.65
   664.7 2389.16   681.4 2395.21   706.4 2406.83   752.4 2425.62793.9377 2444.17
#Mann= 11 ,-1,0
       0     .06       0      90     .05       0     160     .06       0
     200     .05       0     310     .06       0     420     .05       0
   499.2    .045       0   522.7     .05       0     530      .1       0
     580     .06       0     640      .1       0
#XS Ineff= 2 , 0
          483.76 2374.82
Permanent Ineff=
       F       F
Bank Sta=499.2,522.7
XS Rating Curve= 0 ,0
Exp/Cntr(USF)=0,0
Exp/Cntr=0.3,0.1

Type RM Length L Ch R = 1 ,4658    ,459,456.9,455
XS GIS Cut Line= 3
2256125.65047342391038.9096319392255558.86845251391302.942330868
2255376.76431515391477.214579022
#Sta/Elev= 30
       0 2378.86       6 2379.09    23.7  2377.7    41.3 2370.29    45.8  2369.2
    50.2 2369.25      60 2370.16   142.8 2368.39   217.9 2367.56   252.7 2368.13
   306.1 2366.95   376.7 2367.51   412.2 2366.87   500.3 2367.87   510.6 2366.96
   522.3 2365.31   535.6 2363.97   545.3  2365.3   548.8 2367.08   556.7  2373.4
   592.9 2392.12     615 2405.04   625.9 2410.34   637.2  2414.4   663.2 2420.45
   717.6 2429.23   795.1 2450.24   809.8 2453.62   849.4 2460.78   877.3 2467.11
#Mann= 7 ,-1,0
       0     .07       0    50.2     .06       0   306.1     .05       0
   412.2     .06       0   510.6      .1       0   522.3    .045       0
   545.3      .1       0
#XS Ineff= 2 , 0
             240 2374.07
Permanent Ineff=
       F       F
Bank Sta=522.3,545.3
XS Rating Curve= 0 ,0
Exp/Cntr=0.3,0.1

Type RM Length L Ch R = 1 ,4202    ,129.9,145.7,156.9
XS GIS Cut Line= 3
2255845.89325065390628.3424821722255349.46675208390905.488564195
2255306.82889331391316.639345218
#Sta/Elev= 30
       0 2377.04    20.3 2376.58    24.9 2374.81    37.2 2366.26    43.2 2363.63
    59.2  2364.5    75.6 2363.59   140.1 2362.99   223.3 2362.84   249.3 2363.56
   304.7 2362.54   425.2 2362.92     469 2363.52   487.6 2364.61   495.8 2363.61
   501.3 2361.85   505.9 2361.17   521.22361.941   526.9  2364.1   533.4 2367.97
     538 2369.88   559.7 2375.82   628.6 2381.46   640.6 2383.41   693.3 2394.74
   733.1 2401.76   773.1 2405.57   857.3 2411.57   903.3 2415.69   981.9 2424.74
#Mann= 9 ,-1,0
       0     .06       0     110     .05       0     220     .06       0
     280     .05       0     330      .1       0   501.3    .045       0
   521.2      .1       0     560     .05       0  728.55      .1       0
#XS Ineff= 2 , 0
          236.95  2370.9
Permanent Ineff=
       F       F
Bank Sta=501.3,521.2
XS Rating Curve= 0 ,0
Exp/Cntr(USF)=0,0
Exp/Cntr=0.3,0.1

Type RM Length L Ch R = 1 ,4056    ,92.4,85.3,79
XS GIS Cut Line= 4
2255795.73064629390589.9987833212255534.42076115390733.210994542
2255302.09917671390736.8181597642255199.66784266390830.196085447
#Sta/Elev= 30
       0 2376.65       5 2375.91     8.6 2374.01    22.3 2365.06    26.9 2363.76
    37.4  2364.6    63.9 2363.13   154.6 2362.14     198 2362.27   231.8 2363.19
   237.7 2363.05   245.8 2362.14   259.5 2362.62   281.3 2362.25   396.2 2362.68
   406.5 2361.53   416.2 2359.83   428.2 2359.92   432.2 2360.39   436.2 2361.48
   440.2 2362.95   464.2 2365.34   481.4 2369.73   488.2 2370.96   496.3 2371.69
   536.8 2373.08   608.1 2374.19   631.8 2374.06     652 2372.72   668.9 2372.64
#Mann= 7 ,-1,0
       0     .06       0      50     .05       0     160     .06       0
   406.5    .045       0   436.2     .06       0  570.33      .1       0
  590.33     .05       0
Bank Sta=406.5,436.2
XS Rating Curve= 0 ,0
Exp/Cntr=0.5,0.3

Type RM Length L Ch R = 1 ,3970    ,37.2,37.8,36.6
XS GIS Cut Line= 4
 2255695.4685674390452.7100815542255486.39052524390629.279037897
2255268.38842029390700.034107045 2255156.8376356390779.713238968
#Sta/Elev= 30
       0 2376.91     4.3 2376.82     8.3 2376.09    25.5 2366.43    31.7 2363.99
    44.1 2361.92    75.1  2362.1   150.9 2361.18   161.9 2360.72   217.7 2361.34
   229.7 2362.19   239.9 2362.03   249.6 2361.19   267.3 2361.65   305.4 2361.51
     323 2362.22   326.5 2361.99   332.5 2360.29   338.8  2358.9   347.5 2358.81
   354.7 2359.21   360.1 2360.47   368.5 2360.91   381.1 2364.02   385.3 2364.31
   420.5 2364.42   478.5 2367.43   515.3 2368.02   614.9 2371.05639.9428 2371.12
#Mann= 8 ,-1,0
       0     .06       0     180     .07       0  303.66     .06       0
   332.5    .045       0   360.1     .06       0  512.86      .1       0
  612.86     .05       0  632.86      .1       0
#XS Ineff= 2 , 0
          322.92  2365.5  379.72            2366
Permanent Ineff=
       F       F
Bank Sta=332.5,360.1
XS Rating Curve= 0 ,0
Exp/Cntr(USF)=0,0
Exp/Cntr=0.5,0.3

Type RM Length L Ch R = 1 ,3932    ,143.8,145.7,150.9
XS GIS Cut Line= 4
2255649.57338741390406.1774685112255448.78197497 390602.50684957
 2255245.4408303390670.7121864972255136.43977783390755.490782863
#Sta/Elev= 30
       0 2376.09    15.7 2365.55    18.7 2364.02    22.9 2363.23    82.3  2362.1
   124.4    2360     181 2360.68   201.1 2361.62   208.9 2360.35   220.9 2361.33
   246.4 2361.28     256 2360.47   306.8 2361.05   311.8 2359.75   323.7 2358.17
   332.1 2358.92     334  2359.7   340.5 2362.53     349 2363.62   386.9 2363.25
   424.9 2365.22   431.9 2364.64   475.5  2365.7   495.3 2365.14   512.3 2367.29
   531.9 2366.03   537.9 2366.74     558 2365.96   609.1  2368.5633.3889 2368.99
#Mann= 8 ,-1,0
       0     .06       0     130      .1       0     230     .07       0
     270     .06       0   311.8    .045       0     334     .06       0
  380.82     .05       0  480.82      .1       0
#XS Ineff= 3 ,-1
       0      75    2366      75     302  2365.5     337     450    2366
Permanent Ineff=
       F       F       F
Bank Sta=311.8,334
XS Rating Curve= 0 ,0
Exp/Cntr(USF)=0,0
Exp/Cntr=0.5,0.3

Type RM Length L Ch R = 1 ,3787    ,445.8,428.7,412.7
XS GIS Cut Line= 4
2255633.98087554390366.4158525722255521.18556264390450.745708426
2255279.18674756 390495.095694452255070.98227271390728.595143326
#Sta/Elev= 30
       0 2377.44     7.2 2377.18    11.8 2376.38    27.2 2365.56    31.8 2363.17
      38 2361.86    62.2 2361.11   122.1  2360.4   137.1 2359.44   186.6 2360.25
   202.9 2359.46     211 2358.42   219.1 2359.39   227.3 2359.11   231.3  2358.4
   235.4 2357.38   239.5 2357.29   251.7 2357.69   253.8  2358.5   259.8 2360.73
   267.9  2361.3   288.4 2360.24   304.5 2360.12   427.3 2362.25   457.5 2363.74
     529 2364.85   574.6 2366.89   630.8 2367.74   679.1 2369.86   699.7 2370.16
#Mann= 8 ,-1,0
       0     .06       0     100      .1       0  210.83     .05       0
  230.83      .1       0   231.3    .045       0   253.8      .1       0
  310.83     .05       0  616.86      .1       0
#XS Ineff= 2 , 0
                          332.43         2367.37
Permanent Ineff=
       F       F
Bank Sta=231.3,253.8
XS Rating Curve= 0 ,0
Exp/Cntr=0.3,0.1

Type RM Length L Ch R = 1 ,3358    ,685.8,680.5,669.5
XS GIS Cut Line= 4
2255363.90821191390014.0842891612255216.92441637390118.251466336
2254947.86480167390451.7554580252254823.08257084 390613.95171827
#Sta/Elev= 30
       0 2380.99     4.6 2380.01    14.4 2374.17    24.2 2372.73    95.3 2369.34
   122.2 2369.15   185.6 2366.77   240.4 2366.02   245.6 2364.75   255.9 2359.42
   270.5 2355.21   281.6 2355.62   291.8 2355.03   305.1  2355.5   310.8 2356.39
     325 2356.13   378.8 2358.83   389.5 2358.33   461.4 2360.34   506.2 2360.49
   538.1  2361.9   566.8 2361.35   610.5 2363.03   646.5 2362.88   706.3  2364.8
     715 2366.22   739.4 2374.24   752.1 2377.28   794.9 2396.76   813.3 2406.26
#Mann= 7 ,-1,0
       0     .06       0     110      .1       0     130     .06       0
  250.15     .08       0   281.6    .045       0   305.1     .08       0
  580.15      .1       0
#XS Ineff= 2 , 0
                          418.52         2363.59
Permanent Ineff=
       F       F
Bank Sta=281.6,305.1
XS Rating Curve= 0 ,0
Exp/Cntr=0.3,0.1

Type RM Length L Ch R = 1 ,2678    ,465.9,501.1,527.9
XS GIS Cut Line= 4
2255176.46752268389680.3881780652254708.00820447389933.442982633
2254574.31076872390289.8531320482254483.04348573390386.689259369
#Sta/Elev= 30
       0 2371.14     9.7 2370.91    18.5 2368.19    27.6  2367.6   354.9 2358.81
   414.1 2358.31   445.9 2356.44   509.5 2354.53   609.8 2353.54     656  2352.1
   707.3 2353.96   728.7 2352.32   732.9 2350.08   737.2 2348.46   741.5 2348.24
   752.7 2348.51   758.9 2350.11   784.2 2351.01   796.2 2349.78   808.6 2353.57
   814.1 2354.56   886.3 2355.64   895.6 2356.11   903.8 2357.58   913.1 2360.78
   927.9 2368.27   986.2 2402.84  1010.3 2415.93    1027 2423.44  1046.2 2429.66
#Mann= 6 ,-1,0
       0     .06       0      20     .05       0  682.44     .08       0
   732.9    .045       0   758.9     .08       0  892.44      .1       0
Bank Sta=732.9,758.9
XS Rating Curve= 0 ,0
Exp/Cntr=0.3,0.1

Type RM Length L Ch R = 1 ,2176    ,350.7,357.6,364.3
XS GIS Cut Line= 3
2255141.11220447389626.9731211912254662.58518144389814.217464681
2254198.00971563389757.968709658
#Sta/Elev= 30
       0 2368.71    18.2 2366.14    64.2  2364.4   116.7 2363.72     163 2362.47
     190 2361.05   314.6 2358.69   426.2 2355.38     520 2353.98   625.1 2350.34
   662.1 2350.36   673.4 2349.14   709.7 2347.29   725.8 2347.15   737.9 2347.84
     750 2346.42   755.4 2345.17   761.4 2344.79   778.2 2344.84   782.2 2345.31
   794.3 2348.39   798.3 2350.16   802.4 2353.18   810.4 2363.64   814.4 2367.98
   846.7 2393.69   907.1 2438.61   939.4 2465.34   955.5 2477.65   981.8 2500.66
#Mann= 4 ,-1,0
       0     .05       0  703.86      .1       0   755.4    .045       0
   782.2      .1       0
Bank Sta=755.4,782.2
XS Rating Curve= 0 ,0
Exp/Cntr=0.3,0.1

Type RM Length L Ch R = 1 ,1819    ,338.9,353.5,367.6
XS GIS Cut Line= 3
2255117.78371335389610.6949893352254807.22728883389580.744869786
2254356.43796499389380.002301166
#Sta/Elev= 30
       0 2365.83    25.7  2365.1    57.9 2362.94   174.4 2359.77   218.6 2357.11
   263.1  2355.3   481.7 2350.02   510.9 2348.02   564.9 2348.26   578.1 2347.58
   595.6 2345.86   617.5  2346.9   626.2 2345.21   639.4 2344.77   659.4 2342.98
   665.6 2341.93   671.5 2341.69   683.1 2341.88   684.6    2343   687.5 2346.29
   691.9 2354.36   695.7 2359.58     705 2368.78   714.1 2375.37   744.4 2404.27
     762 2419.18   771.4 2428.43   780.5 2436.71   792.7 2446.92   805.5  2458.5
#Mann= 6 ,-1,0
       0     .05       0     352     .06       0     462     .05       0
     572      .1       0   659.4    .045       0   684.6      .1       0
Bank Sta=659.4,684.6
XS Rating Curve= 0 ,0
Exp/Cntr=0.3,0.1

Type RM Length L Ch R = 1 ,1465    ,145.5,147.5,149.8
XS GIS Cut Line= 4
2255033.23600047389579.809191057 2254838.9262747389378.302808777
2254596.63883886388994.4811282422254531.53248658388987.544870754
#Sta/Elev= 30
       0 2362.05    75.9 2361.28   107.3 2363.13   158.2 2359.53     178 2357.27
   203.7 2352.55     237 2349.44   371.1 2346.88   390.2 2345.67   413.2 2342.61
   459.6  2343.1   470.5 2341.59   494.9 2341.43   509.9 2339.83   524.9 2340.66
  528.76 2341.74   536.7 2345.24   541.4 2345.97   645.5 2343.51   683.3 2344.34
   697.5 2343.84   725.9 2345.33   738.3 2346.88   750.4 2346.95   754.4 2347.89
   758.4 2350.92   762.5 2354.88   774.5 2368.49   790.6 2381.36799.3021 2386.57
#Mann= 7 ,-1,0
       0     .06       0     100     .05       0  399.93      .1       0
   494.9    .045       0  528.76      .1       0  629.93     .05       0
  763.83      .1       0
#XS Ineff= 2 , 0
                          541.89         2361.68
Permanent Ineff=
       F       F
Bank Sta=494.9,528.76
XS Rating Curve= 0 ,0
Exp/Cntr(USF)=0,0
Exp/Cntr=0.5,0.3

Type RM Length L Ch R = 1 ,1318    ,76.1,76.1,78.8
XS GIS Cut Line= 3
2255090.60194146389584.8142731572254750.75982849388935.782473087
2254505.54042148388929.118902244
#Sta/Elev= 30
       0 2364.44    40.2 2363.31    87.5 2365.62     126 2365.28   200.1 2359.87
   211.8 2357.21   220.8 2356.81   238.9 2350.94   255.3 2347.17   263.9 2346.26
   416.4 2345.19     433 2341.61   442.1 2340.86   487.5 2341.64   536.9 2339.78
   545.9 2339.27   570.5 2340.23   577.5 2341.45   591.1 2347.44   595.6 2347.83
   600.1 2347.54   609.1 2343.75     615 2342.59   667.8 2341.62   839.2 2342.22
   883.3 2343.92   915.3 2348.34   935.3 2364.67   962.9 2379.83977.9319 2385.86
#Mann= 8 ,-1,0
       0     .05       0      10     .06       0     480      .1       0
   536.9    .045       0   570.5     .05       0     680     .06       0
  812.62     .05       0  912.62      .1       0
#XS Ineff= 2 , 0
          514.15  2351.6  581.13          2350.8
Permanent Ineff=
       F       F
Bank Sta=536.9,570.5
XS Rating Curve= 0 ,0
Exp/Cntr(USF)=0,0
Exp/Cntr=0.5,0.3

Type RM Length L Ch R = 1 ,1242    ,220.8,193.4,161.4
XS GIS Cut Line= 3
2255151.90679321389562.1581322922254818.72825108388895.801048031
2254478.88613811388885.139334683
#Sta/Elev= 30
       0    2370    44.1  2373.6    60.2  2371.6    77.1  2372.3   193.4 2364.92
   215.8 2361.34     256 2358.11   276.7 2351.01   310.6 2345.63   425.9 2344.32
   448.3 2340.84   501.4 2341.69   558.1 2340.33   573.5 2339.01   598.7 2340.49
   640.6 2346.31   662.4 2341.89   751.6 2341.63   763.6 2344.18   771.6 2348.65
   779.6 2349.62   799.6 2349.07   811.6    2344   823.6 2341.74   979.7 2343.62
   995.7 2349.64  1023.7 2351.84  1035.7 2354.27  1067.2 2370.361085.019 2376.05
#Mann= 8 ,-1,0
       0     .06       0      90      .1       0     190     .06       0
   558.1    .045       0   598.7     .06       0     630     .05       0
     640     .06       0  895.01     .05       0
#XS Ineff= 2 , 0
          550.18  2351.6  602.07          2350.8
Permanent Ineff=
       F       F
Bank Sta=558.1,598.7
XS Rating Curve= 0 ,0
Exp/Cntr(USF)=0,0
Exp/Cntr=0.5,0.3

Type RM Length L Ch R = 1 ,1048    ,240.7,256.5,263.9
XS GIS Cut Line= 4
2255352.53857884389026.3957088432255145.92166569388897.487018821
2254865.74290841388876.3257796012254459.34981382388875.196894605
#Sta/Elev= 30
       0 2385.77    52.3 2376.09    80.6 2369.19    94.1 2365.14   127.7  2349.7
   141.9 2345.55   273.4  2341.2   329.5  2341.4   342.4 2337.77   353.6 2337.69
   389.7 2340.17   402.1 2339.05   421.8 2337.26   435.7 2339.04   461.9 2341.41
   488.1 2340.46   590.1 2341.47   598.1 2343.05   610.1 2349.35   614.1 2349.47
   634.1 2348.65   666.1 2341.88   802.1 2342.97   818.1 2345.98   830.1 2350.38
   866.1 2352.33   875.9 2353.74   882.1 2355.28   902.1 2366.19   930.9 2374.57
#Mann= 7 ,-1,0
       0      .1       0   402.1    .045       0   435.7     .07       0
  523.53      .1       0  624.51     .06       0  724.51     .05       0
  914.51     .06       0
#XS Ineff= 2 , 0
          324.87 2356.82  466.17         2356.71
Permanent Ineff=
       F       F
Bank Sta=402.1,435.7
XS Rating Curve= 0 ,0
Exp/Cntr=0.3,0.1

Type RM Length L Ch R = 1 ,792     ,301.7,288.3,264.8
XS GIS Cut Line= 4
 2255359.1756584388866.701206947 2255225.4958754388743.140629715
2254828.86211481388571.2437331682254285.52031183388572.997865343
#Sta/Elev= 30
       0 2377.29    25.8 2366.82    49.4 2359.82    62.6 2357.11   140.3  2353.8
   178.7 2350.24   217.1 2345.48   257.6  2342.5   270.7 2340.73   309.9 2339.44
   353.5 2339.91   370.9 2337.23   379.7 2337.85   403.5 2336.03   418.3 2335.19
   443.32335.897   458.6 2336.21   482.6 2338.65     699 2338.72     775 2340.24
     831 2342.18     847 2345.94     895 2344.05     991 2344.96  1054.5 2347.73
  1079.4 2353.34  1106.7  2357.9    1119 2361.13  1138.8 2369.38  1157.7 2378.93
#Mann= 7 ,-1,0
       0      .1       0   403.5    .045       0   443.3      .1       0
  462.04     .05       0  774.32     .06       0  874.32     .05       0
  974.32      .1       0
#XS Ineff= 2 , 0
          350.94 2351.73  552.07         2344.64
Permanent Ineff=
       F       F
Bank Sta=403.5,443.3
XS Rating Curve= 0 ,0
Exp/Cntr=0.3,0.1

Type RM Length L Ch R = 1 ,504     ,275.5,275,255.4
XS GIS Cut Line= 4
2255308.96489519 388420.19154735 2255173.1726762388388.985195009
2254937.79353823388419.1291947972254285.57070219 388563.04957259
#Sta/Elev= 30
       0 2416.61    50.1 2401.29      87 2388.73   119.8 2373.07   136.3 2363.84
   152.4 2353.57   172.6 2344.29   179.7 2335.96   181.9 2334.48   184.7 2333.22
   204.9 2332.81     225 2334.38   240.5 2335.99   305.7 2335.54   317.8 2334.67
   325.8 2336.29     342 2337.22   374.2 2336.43   615.6 2338.15   708.2 2340.78
   788.6 2341.82   804.7 2344.58   840.9 2342.53   885.2 2344.32   921.1 2347.89
   937.5 2348.39   945.5 2350.73   957.6 2358.37  1013.9 2381.681059.006 2403.34
#Mann= 7 ,-1,0
       0      .1       0   181.9    .045       0     225      .1       0
  249.33     .05       0  646.63     .06       0  756.63     .05       0
  856.63      .1       0
#XS Ineff= 2 , 0
                          447.66         2342.29
Permanent Ineff=
       F       F
Bank Sta=181.9,225
XS Rating Curve= 0 ,0
Exp/Cntr(USF)=0,0
Exp/Cntr=0.3,0.1
